--- RSNRN.prj (project) ---

Proj Title=RSNRN
Current Plan=p01
Default Exp/Contr=0,0
English Units
Geom File=g01
Flow File=f01
Plan File=p01
Background Map Layer=Inundation Boundary (01pct Value_0)
Background Map Layer=QC1
BEGIN DESCRIPTION:
----------MODEL BY WOOD PLC 2021----------
Stream Name: Rosen Run
Flood Zone: Enhanced Approximate
Pocahontas County, WV
HEC-RAS Version: RAS 6.1
Vertical Datum: NAVD88
Projection: NAD 1983 StatePlane West Virginia S FIPS 4702 (US Feet)
Terrain: 1-meter LIDAR (FEMA Region III 3DEP collected 2016-2018)
Land Use: 2019 NLCD
Hydrologic Method:
WV SIR2010-5033 regression equations
Model Notes:
Normal depth tie in to North Fork
END DESCRIPTION:
DSS Export Rating Curves= 0
DSS Export Rating Curve Sorted= 0
DSS Export Volume Flow Curves= 0
DXF OffsetX= 0
DXF OffsetY= 0
DXF ScaleX= 0
DXF ScaleY= 0

--- RSNRN.p01 (plan) ---

Plan Title=Floodplain
Program Version=6.10
Short Identifier=Floodplain
Geom File=g01
Flow File=f01
Subcritical Flow
K Sum by GR= 0
Std Step Tol= 0.01
Critical Tol= 0.01
Num of Std Step Trials= 20
Max Error Tol= 0.3
Flow Tol Ratio= 0.001
Split Flow NTrial= 30
Split Flow Tol= 0.02
Split Flow Ratio= 0.02
Log Output Level= 0
Friction Slope Method= 1
Unsteady Friction Slope Method= 2
Unsteady Bridges Friction Slope Method= 1
Parabolic Critical Depth
Global Vel Dist= 0 , 0 , 0
Global Log Level= 0
CheckData=True
Encroach Param=-1 ,0,0, 0
Mapping Interval=1HOUR
Computation Time Step Use Courant=        0
Computation Time Step Use Time Series=    0
Computation Time Step Count To Double=0
Computation Time Step Max Doubling=0
Computation Time Step Max Halving=0
Computation Time Step Residence Courant=0
Run HTab= 0
Run UNet= 0
Run Sediment= 0
Run PostProcess= 0
Run WQNet= 0
Run RASMapper=-1
UNET Theta= 0
UNET Theta Warmup= 0
UNET ZTol= 0
UNET ZSATol= 0
UNET MxIter= 0
UNET Max Iter WO Improvement= 0
UNET MaxInSteps= 0
UNET DtIC= 0
UNET DtMin= 0
UNET MaxCRTS= 0
UNET WFStab= 0
UNET SFStab= 0
UNET WFX= 1
UNET SFX= 1
UNET Gravity=32.174
UNET 1D Methodology=Finite Difference
UNET DSS MLevel= 1
UNET Pardiso=0
UNET DZMax Abort= 0
UNET Use Existing IB Tables= 0
UNET Froude Reduction=False
UNET Froude Limit= 0
UNET Froude Power= 0
UNET D1 Cores= 0
UNET WindReference=Eulerian
UNET WindDragFormulation=Hsu (1988)
UNET D2 Coriolis=0
UNET D2 Cores= 0
UNET D2 Theta= 1
UNET D2 Theta Warmup= 1
UNET D2 Z Tol= 0.01
UNET D2 Volume Tol= 0.01
UNET D2 Max Iterations= 20
UNET D2 Equation= 0
UNET D2 RampUpFraction=0.1
UNET D2 TimeSlices= 1
UNET D2 Turbulence Formulation=Non-Conservative (original)
UNET D2 Eddy Viscosity=0.3
UNET D2 Transverse Eddy Viscosity=0.1
UNET D2 Smagorinsky Mixing=0
UNET D2 BCVolumeCheck=0
UNET D2 Cores=0
UNET D2 SolverType=PARDISO (Direct)
UNET D2 Minimum Iterations= 2147483647
UNET D2 Maximum Iterations= 2147483647
UNET D2 Restart Number= 10
UNET D2 Relaxation Coeff=1.3
UNET D2 SOR Precondition Iterations= 10
UNET D2 ILUT Maximum Fill= 8
UNET D2 ILUT Tolerance=1E-08
UNET D1D2 MaxIter= 0
UNET D1D2 ZTol=0.01
UNET D1D2 QTol=0.1
UNET D1D2 MinQTol=1
Write IC File= 0
Write IC File at Fixed DateTime=0
Write IC File at Sim End=0
Echo Input=False
Echo Parameters=False
Echo Output=False
Write Detailed= 0
HDF Write Warmup=0
HDF Write Time Slices=0
HDF Flush=0
HDF Compression= 1
HDF Chunk Size= 1
HDF Spatial Parts= 1
HDF Use Max Rows=0
HDF Fixed Rows= 1
Calibration Method= 0
Calibration Iterations= 20
Calibration Max Change=0.05
Calibration Tolerance=0.2
Calibration Maximum=1.5
Calibration Minimum=0.5
Calibration Optimization Method= 1
WQ AD Non Conservative
WQ ULTIMATE=-1
WQ Max Comp Step=1HOUR
WQ Output Interval=15MIN
WQ Output Selected Increments= 0
WQ Output face flow=0
WQ Output face velocity=0
WQ Output face area=0
WQ Output face dispersion=0
WQ Output cell volume=0
WQ Output cell surface area=0
WQ Output cell continuity=0
WQ Output cumulative cell continuity=0
WQ Output face conc=0
WQ Output face dconc_dx=0
WQ Output face courant=0
WQ Output face peclet=0
WQ Output face adv mass=0
WQ Output face disp mass=0
WQ Output cell mass=0
WQ Output cell source sink temp=0
WQ Output nsm pathways=0
WQ Output nsm derived pathways=0
WQ Create Restart=0
WQ Fixed Restart=0
WQ System Summary=0
WQ Write To DSS=0
Sorting and Armoring Iterations= 10
XS Update Threshold= 0.02
Bed Roughness Predictor= 0
Hydraulics Update Threshold= 0.02
Energy Slope Method= 1
Volume Change Method= 1
Sediment Retention Method= 0
Sediment TS Multiplier= 1
Warm Up Method= 0
XS Weighting Method= 0
Number of US Weighted Cross Sections= 1
Number of DS Weighted Cross Sections= 1
Upstream XS Weight=0
Main XS Weight=1
Downstream XS Weight=0
Number of DS XS's Weighted with US Boundary= 1
Upstream Boundary Weight= 1
Weight of XSs Associated with US Boundary= 0
Number of US XS's Weighted with DS Boundary= 1
Downstream Boundary Weight= 0.5
Weight of XSs Associated with DS Boundary= 0.5
Percentile Method= 0
Sediment Output Level= 3
Mass or Volume Output= 0
Output Increment Type= 1
Profile and TS Output Increment= 1
Transport Output Increment 1
XS Output Flag= 0
XS Output Increment= 10
Read HDF5 Sediment Hotstart= 0
Sediment Hotstart Type= 0
Write Gradation File= 0
Read Gradation Hotstart= 0
Write HDF5 File= 1
Write Binary Output= 1
Write DSS Sediment File= 0
DSS Sediment Output Type= 1
SV Curve= 0
Specific Gage Flag= 0
Subcell Erosion Methods= 0
Subcell Deposition Methods= 0
Advection Scheme= 1
Matrix Solver= 0
Implicit Weighting Factor= 1
Maximum Outer Loop Convergence Iterations= 5
Convergence Maximum Absolute= 0.001
Convergence RMSE= 0.0001
Grain Fractions Max Abs Error= 0.001
Max Subgrid Regions= 1
Max Subgrid Length Scale= 3.402823E+38
Initial Layer Thickness= 3.402823E+38
Min Layer Thickness= 3.402823E+38
Max Layer Thickness= 3.402823E+38
Number of Layers= 5

--- RSNRN.f01 (steady flow) ---

Flow Title=Flow
Program Version=6.10
Number of Profiles= 6
Profile Names=01pct,10pct,04pct,02pct,0_2pct,01plus
River Rch & RM=RSNRN,Main,15327
     411     214     287     347     578     608
River Rch & RM=RSNRN,Main,14235
     460     241     322     389     646     681
River Rch & RM=RSNRN,Main,13939
     543     287     382     460     760     804
River Rch & RM=RSNRN,Main,12288
     626     332     441     530     873     925
River Rch & RM=RSNRN,Main,9453
     716     382     506     608     996    1060
River Rch & RM=RSNRN,Main,8581
    1050     566     745     891    1450    1550
River Rch & RM=RSNRN,Main,5952
    1180     643     844    1010    1630    1750
River Rch & RM=RSNRN,Main,5379
    1320     719     942    1120    1810    1950
Boundary for River Rch & Prof#=RSNRN,Main            , 1
Up Type= 0
Dn Type= 3
Dn Slope=0.00478
Boundary for River Rch & Prof#=RSNRN,Main            , 2
Up Type= 0
Dn Type= 3
Dn Slope=0.00478
Boundary for River Rch & Prof#=RSNRN,Main            , 3
Up Type= 0
Dn Type= 3
Dn Slope=0.00478
Boundary for River Rch & Prof#=RSNRN,Main            , 4
Up Type= 0
Dn Type= 3
Dn Slope=0.00478
Boundary for River Rch & Prof#=RSNRN,Main            , 5
Up Type= 0
Dn Type= 3
Dn Slope=0.00478
Boundary for River Rch & Prof#=RSNRN,Main            , 6
Up Type= 0
Dn Type= 3
Dn Slope=0.00478
DSS Import GetInterval= 0
DSS Import GetPeak= 0
DSS Import FillOption= 0

--- RSNRN.g01 (geometry) ---

Geom Title=Geometry
Program Version=6.10

River Reach=RSNRN           ,Main
Reach XY= 30
     2308437.344      508297.1162308649.61028228508911.308278697
     2308520.773      509418.591     2308589.101      509951.323
     2308734.702      510154.038  2308611.969314510253.379631942
     2308637.178      510575.323     2308960.912      511335.487
      2308931.83      511489.201      2308826.15      511546.286
     2308702.779      512261.913     2308404.483      512730.175
     2308276.754      513362.104     2307587.496      513960.201
     2307420.004      513989.897     2307010.772       514971.99
      2306663.95      515084.416     2306442.119       515397.67
     2306471.532      515604.133     2306070.282      515948.925
     2304841.374      515781.577     2304153.555      515481.175
     2304024.754      515639.383     2303964.455      515461.189
     2303447.513      515839.399     2303289.946       516138.62
     2302583.349      516307.215     2302457.717      516154.141
2302117.14541607516099.351608043     2301708.847      516492.339

Type RM Length L Ch R = 1 ,15327   ,324,324,324
XS GIS Cut Line= 4
2308255.84210298508242.9958941762308382.61698675508321.801903006
2308609.89808467508247.564358456 2308722.9675756508192.742787097
#Sta/Elev= 30
       0 2767.28    42.8 2756.81    71.5 2748.49   115.1 2734.79     147 2727.27
     157 2726.16     172 2723.33   197.2 2723.31   205.6 2722.26   209.8 2721.26
     214  2721.1   222.4 2722.24   228.6 2723.19   264.5 2722.59     293 2722.73
   309.6  2725.5   327.6 2727.43   331.9 2729.33   336.1 2731.94   340.3  2732.7
   357.1 2732.16   361.3 2732.45   365.5 2734.96   373.9 2741.03   391.9 2750.03
     414  2762.3   451.7 2780.62   475.4 2790.85     502 2804.49     514 2809.82
#Mann= 8 ,-1,0
       0      .1       0      80     .12       0  189.27      .1       0
   205.6    .045       0   222.4      .1       0  289.27     .06       0
  398.37     .08       0  508.37     .12       0
Bank Sta=205.6,222.4
XS Rating Curve= 0 ,0
Exp/Cntr(USF)=0,0
Exp/Cntr=0.3,0.1

Type RM Length L Ch R = 1 ,15003   ,272.1,283,284.6
XS GIS Cut Line= 3
2308399.74872779508629.0311258332308612.18231681508578.778018753
2308784.64184338508469.134876034
#Sta/Elev= 30
       0    2771      21 2760.26    29.2 2757.36    40.1 2751.54    62.1 2741.45
    70.3  2736.6    82.6 2732.23    86.8 2730.07   103.2 2719.68   107.3 2718.75
  145.512716.805   152.5 2715.95   156.6  2716.8   160.7 2717.68   181.3 2717.22
   218.3 2718.82     242 2719.71   251.3 2721.46   257.1    2722   317.8 2722.69
   320.9 2723.07   332.5 2726.23   341.5 2729.82   346.3 2731.11   365.2 2731.06
   370.1 2732.92   377.8  2737.1   387.5 2741.42   408.3  2747.2   422.7 2751.96
#Mann= 6 ,-1,0
       0      .1       0  145.51    .045       0   156.6      .1       0
   218.3     .05       0   228.3     .06       0   408.3     .08       0
Bank Sta=145.51,156.6
XS Rating Curve= 0 ,0
Exp/Cntr(USF)=0,0
Exp/Cntr=0.3,0.1

Type RM Length L Ch R = 1 ,14720   ,463.2,485.8,473.2
XS GIS Cut Line= 4
2308396.32237958508798.0643041912308536.80265619508841.464714851
2308717.25699525508847.1752952012308963.95406637508677.000000772
#Sta/Elev= 30
       0 2771.27    40.8 2761.68    69.5 2752.29    82.3 2749.28   104.5  2745.3
   125.4 2738.93   142.2 2730.24   150.4 2725.01   165.5 2716.73   170.4  2714.9
   174.4 2714.13   198.4 2714.17   210.4 2713.27   222.4 2713.92   230.4 2712.69
   238.4 2711.29     250 2712.75   258.5 2713.81   266.5 2713.75   314.5 2716.64
     357 2718.22   462.3 2719.86   503.7 2721.17   519.2 2722.29   526.7 2723.42
   535.2 2726.73   542.4 2728.32   563.6 2728.94   578.9 2737.36   627.3 2752.34
#Mann= 6 ,-1,0
       0     .12       0   230.4    .045       0     250     .12       0
  327.03     .08       0  447.58     .05       0  467.58     .06       0
Bank Sta=230.4,250
XS Rating Curve= 0 ,0
Exp/Cntr(USF)=0,0
Exp/Cntr=0.3,0.1

Type RM Length L Ch R = 1 ,14235   ,301.6,296,289.7
XS GIS Cut Line= 3
2308397.83773661509188.1944197252308713.32488803509239.973402652
2308890.36071232509196.106118757
#Sta/Elev= 30
       0 2718.62    14.5 2717.43    22.6 2716.11    30.7 2715.16    34.8 2715.06
      47 2713.23    55.1 2712.36    63.2  2710.6    67.2 2710.07    83.4 2709.59
   103.7 2709.56   115.9 2707.17     124 2706.39   131.7 2706.59   144.2 2706.34
   160.5  2707.2   168.6 2708.49   176.7 2708.64   180.7 2709.15     205 2709.34
   241.5 2711.03   261.8 2710.86   278.1 2711.53   290.2 2712.44   310.4 2714.67
   339.1 2715.91   384.5 2716.86   442.2 2717.55   483.4 2718.88   502.1 2719.19
#Mann= 5 ,-1,0
       0      .1       0      20     .12       0   115.9    .045       0
   160.5      .1       0     220     .05       0
Bank Sta=115.9,160.5
XS Rating Curve= 0 ,0
Exp/Cntr(USF)=0,0
Exp/Cntr=0.3,0.1

Type RM Length L Ch R = 1 ,13939   ,91.7,92.1,92.9
XS GIS Cut Line= 4
2308327.33005526509451.8006497192308467.35476047509511.010549578
2308643.79067798509489.4929867312308743.18140977509454.574315414
#Sta/Elev= 30
       0 2718.53    26.1 2715.88      40 2714.03      53 2712.74      78  2712.2
   126.8 2709.75   135.5 2708.84   160.9 2707.11   181.1 2706.17   189.1 2703.58
   193.2 2703.21   205.2 2704.43   213.3 2704.46   217.3 2703.55   219.7 2702.55
   221.4 2701.85   226.2 2700.92   233.5  2701.2   238.1 2702.35   253.6 2705.68
   257.6 2705.84   269.7 2705.61   281.8 2706.64   293.9 2706.18     306 2706.51
   322.1 2706.25   342.9 2706.91   372.6 2707.33   389.5 2708.21   435.1  2711.6
#Mann= 4 ,-1,0
       0      .1       0   219.7    .045       0   238.1      .1       0
  302.03     .05       0
Bank Sta=219.7,238.1
XS Rating Curve= 0 ,0
Exp/Cntr(USF)=0,0
Exp/Cntr=0.3,0.1

Type RM Length L Ch R = 1 ,13847   ,58.9,58.3,58.3
BEGIN DESCRIPTION:
structure xs 4
END DESCRIPTION:
XS GIS Cut Line= 2
2308194.90495647509620.0322445972308763.14295179509577.731649412
#Sta/Elev= 30
       0 2716.09    21.3 2714.33      30    2714    65.5 2712.62   117.6 2712.11
   133.6 2711.12   145.7 2711.28   157.7 2710.69   213.9  2709.6   237.9 2708.59
   246.5 2708.82     262 2707.89   294.1  2704.4   326.2 2703.05   330.2 2702.64
   334.2 2701.55   342.2 2700.84   354.2 2699.79   361.7 2699.66   366.3 2699.73
   370.3 2700.78   374.3 2703.12   378.3  2703.9   402.4 2703.48   410.4 2703.97
   426.4 2703.64   450.5 2704.23   466.6 2705.31   542.8 2707.27   569.8 2709.38
#Mann= 5 ,-1,0
       0     .12       0      30      .1       0     320     .06       0
   342.2    .045       0   370.3     .06       0
Bank Sta=342.2,370.3
XS Rating Curve= 0 ,0
Exp/Cntr(USF)=0,0
Exp/Cntr=0.5,0.3

Type RM Length L Ch R = 1 ,13788   ,33.8,33.9,33.9
BEGIN DESCRIPTION:
structure xs 3; 11.8 ft between structure and xs
END DESCRIPTION:
XS GIS Cut Line= 2
2308269.22131797509672.4540836572308793.01162308509634.237623627
#Sta/Elev= 30
       0 2715.55      11 2714.02      27 2712.76    39.1 2711.48    51.1 2710.84
   111.2 2709.19   155.4 2708.59     190 2706.91   207.7 2705.58     216 2705.64
   227.6 2705.06   235.6 2705.13   243.6 2704.57   251.6 2703.29     275 2702.16
   280.9 2701.01   283.7 2700.01   287.7 2699.18   291.7  2699.2   295.7 2699.77
   299.7 2700.96   303.8 2702.53   307.8 2703.11   354.4 2703.19   387.1 2704.57
   416.1 2705.26   484.3 2705.81   504.3  2707.2   516.3 2708.55   525.2 2710.03
#Mann= 6 ,-1,0
       0      .1       0     150     .05       0     190      .1       0
     250     .06       0   280.9    .045       0   299.7     .06       0
#XS Ineff= 2 , 0
             269  2703.4311.0103         2703.17
Permanent Ineff=
       F       F
Bank Sta=280.9,299.7
XS Rating Curve= 0 ,0
Exp/Cntr(USF)=0,0
Exp/Cntr=0.5,0.3

Type RM Length L Ch R = 1 ,13754   ,100.9,100,103.3
BEGIN DESCRIPTION:
structure xs 2; 11.6 ft between structure and xs
END DESCRIPTION:
XS GIS Cut Line= 2
2308282.33480915509705.4251472122308806.12511426509667.208687182
#Sta/Elev= 30
       0  2719.1     1.8 2718.55     9.9 2717.17    20.6 2714.51    25.9 2713.53
    37.9 2712.02    46.8 2711.41      58 2710.19   106.1  2709.3   126.2 2708.56
   147.7 2708.28   210.4 2706.46   223.3  2705.7   237.4 2703.51   244.9 2702.67
   266.5 2701.88     270 2700.87   278.6 2699.28   286.6 2699.73   291.6 2700.82
   298.6 2702.33   306.7 2702.81   318.7 2702.42   358.8 2702.51   390.7 2703.69
     430 2704.56   469.2  2704.7   483.1  2705.1   495.4 2706.11   525.2 2710.27
#Mann= 6 ,-1,0
       0      .1       0     140     .05       0     240     .07       0
     270    .045       0   291.6     .07       0     430     .06       0
#XS Ineff= 4 ,-1
       0   258.5  2703.1  303.01308.1502  2702.7308.1502419.2539 2704.09
419.2539   525.2  2702.7
Permanent Ineff=
       F       F       F       F
Bank Sta=270,291.6
XS Rating Curve= 0 ,0
Exp/Cntr(USF)=0,0
Exp/Cntr=0.5,0.3

Type RM Length L Ch R = 1 ,13654   ,139.7,139.5,140.4
BEGIN DESCRIPTION:
structure xs 1
END DESCRIPTION:
XS GIS Cut Line= 3
2308256.94582941509813.2049626082308658.80148366509776.544446781
2308805.75952195 509713.11339324
#Sta/Elev= 30
       0 2740.05    23.3 2730.25    63.5  2715.8    88.3 2709.57    91.6 2709.22
   119.7 2707.89   143.8 2707.46     180  2707.6   220.2 2706.37   244.2 2705.03
   264.3 2702.88   284.4 2702.56   292.4 2701.79   300.5 2701.84   304.5 2701.55
   315.9 2699.95   320.6 2698.98   324.6 2698.91   332.6  2699.3   348.7 2699.28
   352.7    2700   360.7 2700.79   372.8 2701.12   379.2 2701.61   396.8 2701.28
   409.4  2701.4   452.9 2703.44   535.7 2705.48   548.8 2706.12   563.6 2707.38
#Mann= 6 ,-1,0
       0      .1       0      60     .05       0     260     .07       0
   315.9    .045       0   352.7     .07       0  463.52     .06       0
Bank Sta=315.9,352.7
XS Rating Curve= 0 ,0
Exp/Cntr(USF)=0,0
Exp/Cntr=0.3,0.1

Type RM Length L Ch R = 1 ,13515   ,285.1,289.5,286.9
XS GIS Cut Line= 3
2308316.82105982509873.0415774332308537.58171557509927.955282286
2308812.55426988509900.930929062
#Sta/Elev= 30
       0 2720.76    24.1 2713.57    32.3 2711.23    35.9 2710.44    40.6 2709.49
    44.7 2708.99    65.3 2706.97      90 2705.77   139.5 2705.13     156 2704.62
   172.5 2704.41   209.6  2703.5     226 2702.73   234.1 2702.59   250.2 2700.06
     258 2699.58   262.2 2699.09   266.3 2699.08   274.3 2698.76   283.6 2699.09
   294.4 2699.12   302.4 2698.85   314.5 2699.41   334.3  2699.4   346.7 2700.01
   358.7 2699.78   370.8 2700.08   394.9 2699.97   451.2 2701.18   503.8 2702.98
#Mann= 6 ,-1,0
       0      .1       0     110     .05       0     210     .07       0
   266.3    .045       0   283.6     .07       0  503.79     .03       0
Bank Sta=266.3,283.6
XS Rating Curve= 0 ,0
Exp/Cntr(USF)=0,0
Exp/Cntr=0.3,0.1

Type RM Length L Ch R = 1 ,13225   ,182.7,182.6,179.2
XS GIS Cut Line= 3
2308298.60510742 510143.008433122308836.14130874510164.112625781
 2309019.8719272510110.731432579
#Sta/Elev= 30
       0 2726.86    13.6 2721.69    37.6  2716.7    65.6 2707.59    77.6 2705.79
   101.6  2703.8   125.7 2702.82   169.7 2702.12   253.8 2699.47   277.8 2699.78
   293.8 2697.82   301.8 2696.21   313.8 2695.05   325.8 2697.54   329.8 2697.97
   337.8 2696.69   349.8 2695.93   365.9 2696.16   377.9 2695.65   409.9 2696.19
   421.9 2695.72   441.9 2695.69   465.9 2696.19   481.9 2698.32     498 2699.48
   571.3 2700.96   625.5 2703.14   675.4 2706.57   700.4 2708.87   729.3 2709.92
#Mann= 7 ,-1,0
       0      .1       0     220     .05       0     320     .07       0
     420     .08       0   421.9    .045       0   441.9     .08       0
  617.95     .05       0
Bank Sta=421.9,441.9
XS Rating Curve= 0 ,0
Exp/Cntr(USF)=0,0
Exp/Cntr=0.3,0.1

Type RM Length L Ch R = 1 ,13043   ,198.3,200.7,195.6
XS GIS Cut Line= 2
2308330.26686106510260.1812517292309169.22866556510264.411311247
#Sta/Elev= 30
       0 2717.29    13.9 2712.81    25.9 2710.23    57.9 2706.42   137.9 2702.16
   213.9 2699.09   226.1 2699.23   253.9 2696.72   265.9 2696.51   269.9 2695.47
   278.3 2694.89   290.4 2695.48   297.9 2696.17   309.9 2694.92   325.9 2694.85
   337.9 2695.48   382.8 2695.23   405.9 2696.35   417.9 2697.83   529.9 2699.22
   609.9 2702.03   661.9 2706.85   701.9 2709.52   721.9 2712.08   753.9 2714.63
   761.9 2714.17   785.9 2714.81   793.9 2720.65   797.9 2722.57     839 2727.46
#Mann= 7 ,-1,0
       0      .1       0      90     .05       0   269.9    .045       0
   290.4     .07       0     380     .08       0     480     .05       0
     780     .07       0
Bank Sta=269.9,290.4
XS Rating Curve= 0 ,0
Exp/Cntr(USF)=0,0
Exp/Cntr=0.3,0.1

Type RM Length L Ch R = 1 ,12842   ,150.4,151.8,152
XS GIS Cut Line= 4
2308353.93099048 510337.746020512308567.17473164510418.691603889
2308725.58436793510393.450507997 2309092.8858323 510291.61574181
#Sta/Elev= 30
       0 2708.37    32.3 2706.66    49.5 2706.16   143.6 2701.65   199.2 2699.41
   228.1 2697.22   240.8 2694.57   245.3 2694.17   294.9 2694.23   303.7 2694.22
     314 2694.01   322.3 2693.06   330.4  2692.6   342.1 2692.94   362.8  2692.8
   366.8 2692.96   370.9 2694.01   387.1 2694.77   414.8 2694.88   446.1 2696.16
   506.7  2697.2   544.8 2698.65   557.2 2699.43   569.7 2699.41   598.6 2700.46
   683.3 2707.07   731.6 2712.73   752.3 2713.88   764.8 2713.44   769.7 2713.89
#Mann= 6 ,-1,0
       0      .1       0      70     .05       0     170     .07       0
   294.9    .045       0   303.7     .07       0   478.5     .05       0
#XS Ineff= 2 , 0
                          394.68         2697.58
Permanent Ineff=
       F       F
Bank Sta=294.9,303.7
XS Rating Curve= 0 ,0
Exp/Cntr(USF)=0,0
Exp/Cntr=0.3,0.1

Type RM Length L Ch R = 1 ,12690   ,282.2,281.3,274
XS GIS Cut Line= 4
2308369.74741657510563.3355172212308668.67162254510552.055358505
2308718.20611445510551.4366322732308943.20915503510417.336752633
#Sta/Elev= 30
       0 2711.16    18.4 2704.99    26.4 2702.83    30.4 2702.48    50.5 2701.18
     124 2699.52     150 2698.22   178.6  2694.7   186.6 2694.29   214.6 2693.72
   250.6 2693.84   254.6  2693.2   258.2 2690.53   262.6 2689.23   266.6 2689.28
   274.4 2690.53   282.1 2691.16   294.6 2690.24   298.6 2690.93   310.6 2690.86
   330.6 2689.49   338.6 2691.82   342.6  2692.2   351.8 2691.69     413 2692.76
   445.1 2694.93   518.1 2696.97   558.9 2699.07     591 2699.86   610.6 2701.18
#Mann= 9 ,-1,0
       0     .05       0      50     .06       0     150     .05       0
     250     .07       0   258.2    .045       0   274.4     .07       0
  348.68     .08       0  368.68     .07       0  458.68     .05       0
#XS Ineff= 2 , 0
                          345.35         2695.95
Permanent Ineff=
       F       F
Bank Sta=258.2,274.4
XS Rating Curve= 0 ,0
Exp/Cntr(USF)=0,0
Exp/Cntr=0.3,0.1

Type RM Length L Ch R = 1 ,12409   ,124,121.2,112.5
BEGIN DESCRIPTION:
structure xs 4
END DESCRIPTION:
XS GIS Cut Line= 4
2308413.54955907510814.7118205812308603.77716927510796.284758859
2308801.63058393510760.2215626132308999.19169799510561.880397801
#Sta/Elev= 30
       0 2702.67    10.7 2700.11    18.7 2698.87    46.8 2696.22      91 2694.61
   179.2  2693.6   191.5 2692.81     220 2689.04   260.6 2688.45   300.7 2689.15
   305.4 2687.75   309.4 2686.74   324.8 2687.05   329.8 2687.81   341.9 2687.97
   354.2 2689.33   362.6 2689.61   404.7 2694.02   407.5 2694.09   421.6 2692.72
   441.4 2692.94   449.9 2694.57   464.3 2696.44   486.9 2696.94   503.8 2698.94
   526.2 2700.84   560.3 2702.56   599.9 2705.38   644.9 2707.15   672.2 2707.48
#Mann= 6 ,-1,0
       0      .1       0      10     .05       0  301.12     .07       0
   305.4    .045       0   329.8     .07       0  402.23     .05       0
#XS Ineff= 2 , 0
                           359.3         2693.92
Permanent Ineff=
       F       F
Bank Sta=305.4,329.8
XS Rating Curve= 0 ,0
Exp/Cntr(USF)=0,0
Exp/Cntr=0.5,0.3

Type RM Length L Ch R = 1 ,12288   ,70,68.8,67.9
BEGIN DESCRIPTION:
structure xs 3; 7.1 ft between structure and xs
END DESCRIPTION:
XS GIS Cut Line= 5
2308433.30179829511024.605479286 2308822.0501675510853.620040787
  2308911.351424510770.585539129 2309000.6526805510654.650574548
2309021.01963374510593.549714837
#Sta/Elev= 30
       0  2704.3      25 2699.25    73.1 2696.45    97.9 2695.43   116.8 2695.67
   177.8 2693.42   208.5 2690.99   230.4 2691.68   247.8 2689.83     281 2689.22
   326.5 2689.47   335.6 2688.17338.6396  2687.3   348.4 2685.59   353.8 2685.95
   357.1 2685.61  367.452687.317   374.6 2688.73   384.1 2689.49   483.1 2695.03
   548.4 2697.65   568.2 2697.66   626.6 2699.52   659.5  2701.1   692.2 2703.57
   707.2 2703.64   716.8 2702.39   719.8 2702.55     724 2704.24   757.4  2705.9
#Mann= 8 ,-1,0
       0     .06       0     220     .05       0     310     .06       0
338.6396    .045       0  367.45     .06       0  454.69     .05       0
  544.69     .07       0  586.63     .05       0
#XS Ineff= 2 , 0
        331.5102  2693.9373.5115          2694.5
Permanent Ineff=
       F       F
Bank Sta=338.6396,367.45
XS Rating Curve= 0 ,0
Exp/Cntr(USF)=0,0
Exp/Cntr=0.5,0.3

Type RM Length L Ch R = 1 ,12219   ,227,232.6,230.8
BEGIN DESCRIPTION:
structure xs 2; 8.9 ft between structure and xs
END DESCRIPTION:
XS GIS Cut Line= 6
2308444.79419476511095.7587494122308849.22265134510914.137121849
2308926.25059523510843.0531450682308965.83743663510790.435810665
2309030.86000088510686.0332249052309050.61998681 510638.89261324
#Sta/Elev= 30
       0  2701.4    43.2 2700.33    56.3 2698.14    69.5 2697.75    95.8 2695.36
   113.3 2696.13     144 2694.22   187.9 2692.53     258 2688.43   304.1 2687.88
   328.3 2688.55   332.6 2688.07336.95652686.446   341.3 2685.66   367.6 2685.09
   377.3 2685.57382.75652686.562   387.1 2686.97     394 2688.66   402.7 2691.44
   433.4 2691.36   474.2  2693.5   584.6 2697.92   619.5 2700.45   643.8 2703.42
     666 2703.99   686.5  2705.5   709.2  2705.9   742.3 2705.74   788.1 2706.81
#Mann= 9 ,-1,0
       0     .06       0      80     .05       0     150     .06       0
336.9565    .045       0382.7565     .06       0  558.15     .07       0
     674     .05       0     694     .06       0  786.99     .05       0
#XS Ineff= 2 , 0
           333.9  2693.9   385.7          2694.5
Permanent Ineff=
       F       F
Bank Sta=336.9565,382.7565
XS Rating Curve= 0 ,0
Exp/Cntr(USF)=0,0
Exp/Cntr=0.5,0.3

Type RM Length L Ch R = 1 ,11986   ,368.3,381.1,377.6
BEGIN DESCRIPTION:
structure xs 1
END DESCRIPTION:
XS GIS Cut Line= 2
2308450.11854742511330.3863099072309035.27678081511072.352679279
#Sta/Elev= 30
       0  2706.5    15.4 2705.83    19.7 2703.95    24.1 2701.06    28.5 2699.03
    32.8 2697.72      46 2694.99    59.1 2693.25    85.3 2692.82   146.5    2691
   245.2 2689.39   277.7 2688.51   325.7 2688.74   372.6 2687.62   390.8 2687.64
   395.7 2687.25   400.1 2685.21   404.4 2684.11   408.8 2683.97   423.9 2685.23
   430.2 2685.48   474.4  2684.3   487.9  2685.4   518.5 2685.65   545.5 2685.31
   557.7 2687.43   569.8  2692.8   579.3 2696.15   605.5 2706.29   639.5 2717.53
#Mann= 7 ,-1,0
       0     .06       0      70     .07       0     180     .05       0
     400      .1       0   400.1    .045       0   423.9      .1       0
     610     .12       0
Bank Sta=400.1,423.9
XS Rating Curve= 0 ,0
Exp/Cntr(USF)=0,0
Exp/Cntr=0.3,0.1

Type RM Length L Ch R = 1 ,11605   ,163.4,169.9,167
XS GIS Cut Line= 2
2308421.91815063511438.9578375482309022.58660225 511462.92817482
#Sta/Elev= 30
       0 2708.13    10.3 2708.55    18.3 2708.36    34.3 2706.42    46.3 2703.51
    74.3 2694.88    90.3 2692.24   110.3 2690.41   192.9 2687.39   274.5 2686.41
   306.5 2685.12   394.6 2684.54   410.6  2682.9   434.6 2682.81     447 2681.84
   466.6 2682.41   478.6 2681.31   482.6 2681.31   490.6 2682.32   494.7 2682.07
   498.7 2681.02   502.7 2679.93   506.7 2679.78   522.7  2681.1   542.7 2683.54
   554.7 2684.47   562.5 2687.47   582.7 2696.95   594.7 2701.77   601.1 2703.83
#Mann= 5 ,-1,0
       0     .06       0     100     .05       0     490      .1       0
   498.7    .045       0   522.7      .1       0
Bank Sta=498.7,522.7
XS Rating Curve= 0 ,0
Exp/Cntr(USF)=0,0
Exp/Cntr=0.3,0.1

Type RM Length L Ch R = 1 ,11435   ,200.1,204.4,203.9
XS GIS Cut Line= 4
2308415.29887861511493.6767634512308762.89734597511547.057956653
2309017.38908101511571.8864186082309155.18704485511643.888958276
#Sta/Elev= 30
       0 2708.34    17.1 2708.48    33.3 2706.55    73.7 2694.45    89.9 2691.59
   106.1 2689.83   146.6 2687.88   197.7 2686.73   336.3 2685.38   369.4 2684.37
   397.2 2682.64   401.2 2682.08   405.32680.542   413.2 2679.32   420.7 2680.51
   437.4 2681.93   445.4 2681.17   455.9 2682.58   497.7  2682.5   521.8 2683.53
   561.9 2686.86   590.1 2688.04   627.4 2691.29   644.7 2693.26   653.4 2695.58
   670.6 2698.55   699.3 2701.22   713.8 2703.22     729 2706.46   762.8 2715.48
#Mann= 6 ,-1,0
       0     .06       0     100     .05       0   405.3    .045       0
   420.7     .05       0  501.67      .1       0  707.37     .12       0
Bank Sta=405.3,420.7
XS Rating Curve= 0 ,0
Exp/Cntr(USF)=0,0
Exp/Cntr=0.3,0.1

Type RM Length L Ch R = 1 ,11231   ,335.7,334.5,331.4
XS GIS Cut Line= 4
2308406.98375928511620.4495167312308761.64263401511689.086925034
 2308944.7135091511742.1509467982309042.90270689511688.130469027
#Sta/Elev= 30
       0 2706.76     8.5 2706.06    21.6 2703.99    42.6  2696.5    54.2 2693.31
    66.5 2690.83    82.7 2689.13   172.3 2686.94   305.4 2685.66   339.4 2684.88
   361.6 2684.03   388.9 2682.29     393 2681.73   397.2 2679.65   398.9 2679.34
   402.1 2678.89   413.9 2678.95   417.6 2679.37   433.4 2680.65   451.3 2680.42
     468  2681.7   489.3 2680.82   537.7 2681.73   547.1 2682.38   574.1 2683.04
   592.3 2684.91   603.7 2686.79   628.5 2692.37   651.7 2697.15   663.9 2700.19
#Mann= 8 ,-1,0
       0      .1       0      10     .06       0      40     .07       0
     110     .05       0     310      .1       0   398.9    .045       0
   417.6      .1       0  621.85     .12       0
Bank Sta=398.9,417.6
XS Rating Curve= 0 ,0
Exp/Cntr(USF)=0,0
Exp/Cntr=0.3,0.1

Type RM Length L Ch R = 1 ,10896   ,164.9,162.6,159.9
XS GIS Cut Line= 4
2308355.64721817 511826.713293412308644.70128527512005.785813026
2308816.72370569512025.5260907792309107.18779262511902.854364743
#Sta/Elev= 30
       0 2701.13    19.4 2700.14    24.1 2699.41    28.3 2697.88    33.6 2696.94
    71.2 2693.02   132.4 2689.63   231.7 2685.93   278.2 2681.84   315.9 2680.63
   355.6 2678.71   395.9 2678.05   403.9 2677.41   407.6 2676.28     412 2675.23
     416 2674.93   422.92676.286   444.2 2677.84   472.4 2678.33   500.5  2679.8
   522.2 2679.88   575.8 2683.73   647.3 2686.63   678.6 2687.14   712.3 2689.25
   740.3 2692.74   763.4 2696.45   781.7 2701.09   791.7 2704.17   828.5 2717.18
#Mann= 9 ,-1,0
       0      .1       0      70     .05       0   407.6    .045       0
   422.9     .05       0  510.03      .1       0  533.18     .05       0
  723.18      .1       0  783.18     .05       0  828.49      .1       0
Bank Sta=407.6,422.9
XS Rating Curve= 0 ,0
Exp/Cntr(USF)=0,0
Exp/Cntr=0.3,0.1

Type RM Length L Ch R = 1 ,10734   ,390.1,401.7,415.4
XS GIS Cut Line= 4
2308330.26686106512173.5781739272308611.89126296512184.349665662
2308788.14374289512170.249467267  2309077.577376512221.518848469
#Sta/Elev= 30
       0  2697.3     5.9 2696.03    17.9 2694.41    25.9 2691.67    49.9  2691.7
      58  2691.2      70 2689.32      82 2688.33     146  2684.3   248.2 2679.49
   302.2 2678.81   340.8 2678.89   366.8 2679.56   370.4 2679.37   377.9  2675.8
   390.5 2674.75   394.5 2675.73   398.5 2678.05   402.5 2678.92   410.5 2679.41
   434.6 2678.44   552.1 2681.85   596.8 2684.97   654.5  2689.9     674 2692.37
   682.1 2694.38   690.2 2695.58   706.5 2699.56   730.8 2706.94   752.6 2712.48
#Mann= 4 ,-1,0
       0     .06       0      90     .05       0   377.9    .045       0
   394.5     .05       0
Bank Sta=377.9,394.5
XS Rating Curve= 0 ,0
Exp/Cntr(USF)=0,0
Exp/Cntr=0.3,0.1

Type RM Length L Ch R = 1 ,10332   ,366.1,357.8,348.1
XS GIS Cut Line= 4
2308413.45803159512433.0218243942308496.88484977512476.788028713
2308631.01122931512631.0143368892308967.53484362  512658.7465475
#Sta/Elev= 30
       0 2684.91    12.1 2684.44    16.6 2683.15    21.1 2680.97    25.7 2679.82
    34.7 2679.06      88  2677.4   105.3 2676.31   147.9 2675.16   153.5 2674.44
   159.2 2672.66   163.6 2672.01     179 2671.39   181.9 2672.09   184.8 2673.48
   190.1 2674.23   206.1 2674.52   227.3 2674.03   259.1 2675.33   311.8 2676.31
   339.9 2677.91     360 2678.03   371.9 2679.33   432.2 2681.48   468.5 2683.78
   509.3 2683.88   532.6 2684.49   584.7 2688.45   620.9 2693.55   636.3 2696.45
#Mann= 4 ,-1,0
       0     .06       0      10     .05       0   163.6    .045       0
   181.9     .05       0
Bank Sta=163.6,181.9
XS Rating Curve= 0 ,0
Exp/Cntr(USF)=0,0
Exp/Cntr=0.3,0.1

Type RM Length L Ch R = 1 ,9974    ,308.2,310.5,311.4
XS GIS Cut Line= 3
2308317.53264998512828.6662181622308574.15626077512880.836952224
2309039.30176911512757.165348785
#Sta/Elev= 30
       0  2682.1     2.7 2679.71     6.8  2677.4    14.9 2678.11    27.2 2678.14
    31.3 2677.59    39.4 2673.48    63.7 2672.41    72.1 2670.65    76.2 2669.98
    80.3 2669.88    84.3 2669.93    88.4 2670.56    92.5 2671.28     117 2671.38
   133.3 2672.14   174.1 2672.62   236.7 2676.55   359.2 2680.45   462.7 2684.85
   549.6 2687.57   603.4 2688.09   673.7 2691.91   690.3 2692.33   694.4 2692.75
   702.7 2694.78   707.9 2695.29   717.7 2697.17   731.7 2701.14   743.2 2705.01
#Mann= 5 ,-1,0
       0     .06       0    72.1    .045       0    88.4     .06       0
     100     .05       0  711.87      .1       0
Bank Sta=72.1,88.4
XS Rating Curve= 0 ,0
Exp/Cntr(USF)=0,0
Exp/Cntr=0.3,0.1

Type RM Length L Ch R = 1 ,9664    ,182.8,210.4,219.1
BEGIN DESCRIPTION:
structure xs 4
END DESCRIPTION:
XS GIS Cut Line= 4
2308239.88458935512852.8834320012308296.28538293513132.067360221
2308462.00501466513186.3108234462308771.28172451513197.305038685
#Sta/Elev= 30
       0  2729.1    28.9 2724.26    51.4  2719.2    77.8 2710.77   114.6    2701
   122.7 2697.49     139  2688.1   143.2 2686.18   147.2    2685   151.3 2682.66
   163.5 2677.62   170.2 2675.48     177 2674.47   221.2 2674.05   241.1 2672.86
   269.6 2672.44   297.3 2670.77     310 2668.41   318.4 2667.46   322.6 2667.55
   326.8  2668.4   326.8 2668.41     331 2669.44   390.3 2669.41   444.6 2672.23
   506.6 2673.97   545.6 2676.29   657.7 2679.31   711.6  2681.5   768.7 2682.96
#Mann= 4 ,-1,0
       0     .12       0      60     .06       0     310    .045       0
   326.8     .05       0
Bank Sta=310,326.8
XS Rating Curve= 0 ,0
Exp/Cntr(USF)=0,0
Exp/Cntr=0.5,0.3

Type RM Length L Ch R = 1 ,9453    ,113.1,105.1,104.5
BEGIN DESCRIPTION:
structure xs 3; 15.2 ft between structure and xs
END DESCRIPTION:
XS GIS Cut Line= 6
2308187.99214335512830.6365098172308274.28535752513146.621955847
2308256.51910754513263.3715985572308318.82595989513475.818406885
2308540.77910719513892.8044549062308630.87937493513966.407490527
#Sta/Elev= 30
       0 2743.75      40 2737.41   106.3 2723.67   118.7 2719.53   213.3  2694.9
   256.3 2675.18   262.8 2673.54   301.2 2673.18   334.2 2670.54   463.3 2669.78
   488.8 2668.63   497.1 2667.17   513.6 2667.48   524.8 2666.51  543.832667.599
   552.3 2668.94   573.2 2669.84   589.6 2669.41   602.4 2666.92   671.8 2670.68
   695.9 2670.21   975.4 2673.98  1043.4 2675.84  1061.5 2677.47  1075.1 2677.08
  1106.8 2680.47  1121.8 2680.93  1162.4 2688.08  1203.9  2699.5    1259 2719.13
#Mann= 12 ,-1,0
       0      .1       0     120     .06       0  485.65     .07       0
   513.6    .045       0  543.83     .07       0  596.64     .06       0
  666.64     .05       0  700.28     .08       0  810.28     .06       0
  880.28     .05       0 1030.28     .06       0 1242.66     .12       0
#XS Ineff= 2 , 0
             498  2671.3     558          2672.2
Permanent Ineff=
       F       F
Bank Sta=513.6,543.83
XS Rating Curve= 0 ,0
Exp/Cntr(USF)=0,0
Exp/Cntr=0.5,0.3

Type RM Length L Ch R = 1 ,9348    ,106.1,103.1,110.4
BEGIN DESCRIPTION:
structure xs 2; 18.5 ft between structure and xs
END DESCRIPTION:
XS GIS Cut Line= 6
2308135.32790234512852.8443222892308221.62111652513168.829768319
2308213.17044491 513425.880765882308245.73245577513449.282714394
2308488.11486618513915.0122673782308578.21513393513988.615302999
#Sta/Elev= 30
       0 2733.54    87.4 2711.88   141.3 2695.67   182.8  2684.9   220.1 2678.01
   261.7    2673   303.9 2672.27   332.6 2673.72   388.6 2672.88   445.2 2673.97
   469.3 2669.71   489.6 2671.75   550.9 2671.56   583.1 2666.19   611.2 2665.47
   627.7 2666.16   659.2 2668.39   672.8 2671.04   686.4 2669.32   704.4  2671.7
     763 2670.03  1033.6 2672.59  1101.4 2675.14    1153 2679.38  1163.3  2678.6
  1199.5 2681.42  1209.8 2684.76  1220.1 2685.69  1231.2 2690.59  1269.2 2702.27
#Mann= 16 ,-1,0
       0      .1       0     160     .05       0     260     .06       0
  367.56     .05       0  465.65     .06       0  515.65     .07       0
  540.81     .06       0  560.81     .05       0   583.1    .045       0
   627.7     .06       0  787.87     .08       0  797.87     .06       0
  997.87     .05       0 1017.87     .06       0 1127.87     .05       0
  1192.9     .06       0
#XS Ineff= 2 ,-1
       0576.9818  2671.3  633.98 1269.16  2672.2
Permanent Ineff=
       F       F
Bank Sta=583.1,627.7
XS Rating Curve= 0 ,0
Exp/Cntr(USF)=0,0
Exp/Cntr=0.5,0.3

Type RM Length L Ch R = 1 ,9245    ,385.3,382.4,379.5
BEGIN DESCRIPTION:
structure xs 1
END DESCRIPTION:
XS GIS Cut Line= 3
2308062.36309155513307.2341248812308197.72499615513585.008033262
 2308545.9998965514078.514977086
#Sta/Elev= 30
       0 2686.97    15.5 2685.55    47.7  2685.2    86.7  2681.9    95.6 2680.31
   101.5 2678.16   116.5 2674.79   130.5  2673.5   152.4 2672.44   168.5 2669.43
     205 2668.13   220.2 2665.71     238 2664.79   248.1 2665.68   260.2 2667.85
   300.3 2667.23   310.9  2668.2   434.3  2670.2   519.7  2670.7   569.2 2670.83
   646.7 2671.78   701.7 2674.04   775.9 2678.84   819.7 2683.06   833.5 2682.45
   861.3 2684.75   868.2 2685.19   886.9 2692.16   902.9 2699.76     913 2702.39
#Mann= 8 ,-1,0
       0     .05       0   116.5     .06       0   130.5     .05       0
   220.2    .045       0   248.1     .05       0   519.7     .06       0
   569.2     .05       0   861.3     .06       0
#XS Ineff= 1 ,-1
     320 912.976    2670
Permanent Ineff=
       F
Bank Sta=220.2,248.1
XS Rating Curve= 0 ,0
Exp/Cntr(USF)=0,0
Exp/Cntr=0.3,0.1

Type RM Length L Ch R = 1 ,8863    ,283.7,282.1,280.2
XS GIS Cut Line= 3
2307750.74870703513587.8280729412307901.62082985513809.201187742
  2308194.895662513983.939598982
#Sta/Elev= 30
       0 2682.67    11.3 2679.79    30.7 2676.31    48.1 2674.54    59.6 2673.98
    74.2 2672.32    79.7 2671.53    88.8 2669.61   103.3 2670.55     113 2670.18
   123.3 2670.45   130.4 2669.99   137.2 2668.64   145.9 2665.08   151.7 2664.06
   160.3 2663.31   166.2 2662.46   174.7  2662.2   180.7  2662.6  183.852663.269
   190.4 2664.23   195.3 2664.38   217.9 2664.09   229.8 2664.41   312.8 2664.92
     378 2667.59   430.2 2667.77   517.8 2669.34   541.1 2670.03   609.3 2670.87
#Mann= 4 ,-1,0
       0     .05       0   160.3    .045       0  183.85     .05       0
     250     .07       0
Bank Sta=160.3,183.85
XS Rating Curve= 0 ,0
Exp/Cntr(USF)=0,0
Exp/Cntr=0.3,0.1

Type RM Length L Ch R = 1 ,8581    ,430.7,433.6,431.3
XS GIS Cut Line= 2
2307470.40333945513721.3809005752307813.71046771514121.395009844
#Sta/Elev= 30
       0 2696.53    15.5 2693.13    31.4 2690.68    41.9 2688.57    52.2 2686.25
      72 2681.15    86.2 2675.55    94.7 2673.41    99.9 2673.11   103.2 2672.16
   106.1 2670.85   111.7 2667.47   115.7 2665.94     121 2665.38   150.1 2664.26
   189.5 2663.21   205.4 2663.31   211.5 2662.61   223.8 2662.04     229 2661.45
   242.2 2661.03   248.92661.568     258 2662.23   281.9 2662.32   294.9 2661.99
   305.5 2662.62   328.2 2663.03   389.7  2666.5   469.2 2668.09   527.1 2668.85
#Mann= 5 ,-1,0
       0      .1       0     100     .08       0     229    .045       0
   248.9     .08       0     250     .05       0
Bank Sta=229,248.9
XS Rating Curve= 0 ,0
Exp/Cntr(USF)=0,0
Exp/Cntr=0.3,0.1

Type RM Length L Ch R = 1 ,8147    ,201.9,197.3,192.9
XS GIS Cut Line= 3
2307267.86555023514053.4266045762307481.73113297514251.250491632
2307725.50077812514264.975578965
#Sta/Elev= 30
       0 2683.49      17 2674.75    38.6 2670.27    48.2  2667.8    60.4 2665.64
    76.7 2663.62   103.9 2661.68   114.8 2659.76   123.3 2659.24   135.9  2659.4
   142.1 2657.96   146.9 2657.28   170.5 2656.73   180.2    2656   185.7 2656.29
   186.9 2656.73   189.7 2658.43   191.1 2659.03   192.5 2659.15   226.5 2659.26
   237.8 2659.85     247 2660.99   271.8 2662.47   297.8 2663.51   321.8 2663.65
   349.9 2664.72   377.9 2666.34   486.1 2668.72   514.1 2668.34   535.5 2668.47
#Mann= 6 ,-1,0
       0     .12       0      60      .1       0      90     .08       0
   170.5    .045       0   186.9     .08       0     200     .05       0
Bank Sta=170.5,186.9
XS Rating Curve= 0 ,0
Exp/Cntr(USF)=0,0
Exp/Cntr=0.3,0.1

Type RM Length L Ch R = 1 ,7950    ,280.3,282.1,283.8
XS GIS Cut Line= 3
2307071.92185129514228.678487426 2307442.8161595 514406.46253599
2307637.45904025514407.995157098
#Sta/Elev= 30
       0 2730.36     3.6 2729.67     9.6 2727.04    53.5 2713.62      89 2703.99
   111.2 2697.32   124.5 2691.88   164.4 2673.23   182.1 2668.36   195.5 2666.09
   204.3 2664.12   217.6 2662.56   228.5 2658.81   230.9 2657.71   234.4 2655.48
   235.4 2655.05   241.8 2654.99     251 2655.48   261.4 2655.98   269.5 2657.11
   279.7 2657.69     293 2657.84   342.4 2659.81     364 2660.16   408.3 2662.19
   439.2 2663.05   504.7 2665.77   564.7 2666.34   592.7 2668.22     606 2668.58
#Mann= 5 ,-1,0
       0      .1       0     180     .08       0   234.4    .045       0
     251     .08       0     290     .05       0
Bank Sta=234.4,251
XS Rating Curve= 0 ,0
Exp/Cntr(USF)=0,0
Exp/Cntr=0.3,0.1

Type RM Length L Ch R = 1 ,7668    ,172.9,169.6,167.6
XS GIS Cut Line= 3
2307049.88967957514511.6364703732307366.00911005514701.129333128
2307464.09509607514831.939422512
#Sta/Elev= 30
       0 2750.82    10.8 2741.98    21.3 2732.57    26.3 2728.92    30.6 2726.19
    49.4 2711.34    55.3 2707.17      68 2696.42    72.8 2691.72    81.9 2681.89
    90.3 2673.35      99 2663.55   101.9 2661.14   111.9 2655.73   116.5 2654.13
   119.3 2653.77   135.3 2654.57   147.2 2654.04   165.2 2653.25     169 2653.61
   170.6 2654.12   175.2 2656.75   179.9 2657.46   217.2 2658.06   230.2 2659.31
   259.2  2660.5   343.1 2661.67   423.6 2664.09   468.6 2664.34   532.1 2665.52
#Mann= 4 ,-1,0
       0      .1       0   147.2    .045       0   170.6      .1       0
     220     .05       0
Bank Sta=147.2,170.6
XS Rating Curve= 0 ,0
Exp/Cntr(USF)=0,0
Exp/Cntr=0.3,0.1

Type RM Length L Ch R = 1 ,7498    ,241.5,249.5,255
XS GIS Cut Line= 4
2306918.55688311 514544.860043072307008.48725682514701.884712494
2307260.72582056514791.1738957772307395.46104967515048.110844307
#Sta/Elev= 30
       0  2799.5    54.2    2765    74.1 2750.23    83.5  2745.2    97.2 2735.83
     111 2724.75   121.6 2717.55   129.4 2711.27   138.7  2706.4   166.3 2685.11
   175.5 2679.31     181 2674.64     199 2665.98   214.6 2655.95   231.5 2654.05
   248.5 2654.21   255.4 2652.38   265.5 2651.05   274.7 2652.37   345.8 2657.96
   454.6 2660.85   527.6 2660.42   576.5  2661.4   617.9 2664.24   651.1 2665.46
   658.6 2666.76   672.1 2670.67   694.7  2678.9   708.2 2684.78   738.7 2693.74
#Mann= 6 ,-1,0
       0      .1       0   255.4    .045       0   274.7      .1       0
  320.95     .07       0  420.95     .05       0  658.53      .1       0
Bank Sta=255.4,274.7
XS Rating Curve= 0 ,0
Exp/Cntr(USF)=0,0
Exp/Cntr=0.3,0.1

Type RM Length L Ch R = 1 ,7249    ,333.9,329.7,325.3
XS GIS Cut Line= 4
2306829.76771617514712.986757652 2306907.9313927514870.846731808
2307039.73680801514990.3911782562307231.31444655 515059.35912813
#Sta/Elev= 30
       0  2722.4    13.6 2713.19      27 2703.18    46.7 2689.33    58.7  2681.3
    67.2 2674.61    76.1 2668.55    80.6 2664.61    93.9 2655.23    98.4 2654.15
   107.3 2655.39   134.1 2653.45   156.4 2654.13   167.7 2653.55   198.1 2653.96
   206.3 2653.62   214.8 2651.27   219.7  2650.8   251.1 2651.86   298.7  2650.9
   316.9 2650.46   325.2 2650.91   328.1 2651.66   336.6 2656.99   345.1 2659.47
   350.7 2660.52   374.1 2661.78   469.1 2662.75   541.6 2664.55   557.7 2665.86
#Mann= 5 ,-1,0
       0      .1       0    80.6     .12       0   298.7    .045       0
   325.2     .12       0   336.6     .05       0
#XS Ineff= 2 , 0
        185.1803    2660
Permanent Ineff=
       F       F
Bank Sta=298.7,325.2
XS Rating Curve= 0 ,0
Exp/Cntr(USF)=0,0
Exp/Cntr=0.3,0.1

Type RM Length L Ch R = 1 ,6919    ,171.8,171.8,171.6
XS GIS Cut Line= 4
2306613.59970409514851.6709842042306639.98710568515004.054836426
2306855.41688506 515157.399292532307199.54694038515198.237888705
#Sta/Elev= 30
       0 2717.33    29.9 2711.81    46.2 2707.55    58.4 2705.39    90.8 2697.04
   107.1 2693.93   139.6  2686.7   154.7 2681.78   159.8 2679.14   164.7 2675.12
   179.4 2661.04   187.1 2655.17   191.1 2653.26     204 2649.09214.11852647.942
   224.4 2647.11245.71842647.984   273.2 2648.37   290.4 2649.24   310.5 2649.16
     329 2648.42     365 2648.36   370.9 2648.92   393.7 2652.87   431.9 2655.08
   593.1 2658.16   712.7 2661.96   742.1 2663.94   758.2  2667.2   765.6 2669.53
#Mann= 5 ,-1,0
       0      .1       0      30     .12       0214.1185    .045       0
245.7184     .12       0  274.65     .05       0
Bank Sta=214.1185,245.7184
XS Rating Curve= 0 ,0
Exp/Cntr(USF)=0,0
Exp/Cntr=0.3,0.1

Type RM Length L Ch R = 1 ,6747    ,183.6,186.3,188.5
XS GIS Cut Line= 3
2306502.90504946515119.0268835812306665.04511596515228.102928317
2307077.76528523515262.004942222
#Sta/Elev= 30
       0 2673.07    11.2    2671    25.6 2666.57    54.6 2662.49    59.4 2660.67
    73.8 2653.85    99.9 2645.56   103.3 2644.61     112 2644.34   117.7 2644.56
   123.5 2645.62   126.9 2646.26   131.7 2646.58   155.8 2646.64   160.6 2647.16
   168.7 2648.88   172.5 2649.13   195.6 2648.91   262.8 2649.16   286.9 2650.48
   379.2 2651.92   391.2 2652.38   403.2 2652.34   436.7 2655.42   447.8 2656.07
   470.1 2656.62   503.7 2658.04   535.7 2658.18   556.2 2658.92   609.5 2659.85
#Mann= 4 ,-1,0
       0     .12       0    99.9    .045       0   123.5     .12       0
     170     .05       0
Bank Sta=99.9,123.5
XS Rating Curve= 0 ,0
Exp/Cntr(USF)=0,0
Exp/Cntr=0.3,0.1

Type RM Length L Ch R = 1 ,6561    ,101,98.2,95.8
XS GIS Cut Line= 4
2306414.46015703515166.9436531742306414.46015703515266.167271509
2306680.79723783515511.6151694952306988.91268423515670.024805785
#Sta/Elev= 30
       0 2649.18    14.2 2648.09    26.2 2648.89   121.4  2648.2     145 2646.35
   150.5 2644.39   153.5 2644.07   166.8 2644.31     179 2643.88   188.6 2643.25
   199.5  2643.9   204.9 2645.19   210.3 2645.73   269.6 2644.68   286.6  2646.6
   324.6 2647.48   343.2 2646.86   362.7 2647.31   406.2 2647.07   496.7 2648.38
   524.5 2649.26   551.2 2650.95   564.2  2651.1   569.8 2650.53   582.1 2651.88
   634.4 2653.27   643.3  2654.1   684.9 2659.98   759.2 2674.35   807.9 2680.72
#Mann= 6 ,-1,0
       0      .1       0      10     .05       0     179    .045       0
   199.5     .05       0  581.41      .1       0  801.41     .06       0
Bank Sta=179,199.5
XS Rating Curve= 0 ,0
Exp/Cntr(USF)=0,0
Exp/Cntr=0.3,0.1

Type RM Length L Ch R = 1 ,6463    ,200.7,205.8,205.6
XS GIS Cut Line= 3
2306350.20415987515175.6051851582306399.79030428515395.068448177
2306665.77725759515558.993609439
#Sta/Elev= 30
       0 2648.75    30.3 2648.69    95.9 2647.95   149.2 2648.05   156.8 2647.56
   170.2 2645.97   177.9  2645.5   198.5 2645.01     219 2645.52   248.9 2645.12
   253.6 2644.74258.44412642.839   267.1  2642.5   280.9 2642.84   305.3 2643.56
   340.2 2642.85   366.4 2643.09   385.2 2644.39   394.6 2646.03   399.3 2645.89
   404.1 2645.27   408.7 2645.26   412.9 2645.88   418.1 2646.22   427.2 2646.09
   441.9  2646.6   469.8 2646.67   479.2 2646.96   507.4 2646.78   537.4 2647.08
#Mann= 3 ,0,0
       0     .05       0258.4441    .045       0   280.9     .05       0
#XS Ineff= 1 ,-1
 108.088 224.933    2648
Permanent Ineff=
       F
Bank Sta=258.4441,280.9
XS Rating Curve= 0 ,0
Exp/Cntr(USF)=0,0
Exp/Cntr=0.3,0.1

Type RM Length L Ch R = 1 ,6257    ,184.9,187.8,188.4
XS GIS Cut Line= 4
2306345.78167783515367.9902807112306380.62161979515540.046495927
2306515.58038897515655.5487392632306544.16009037515736.289901873
#Sta/Elev= 30
       0 2645.53    25.7 2644.75    77.7    2645   152.4 2643.65   178.9 2643.85
   193.1 2642.45   206.5 2642.33   211.8  2642.8   215.8 2642.64   222.3 2641.75
   251.1 2641.69   263.4 2640.54   275.7 2640.49   285.5 2640.16  293.58  2640.5
   300.9 2642.29   312.6 2642.24   331.1 2644.08     355 2644.56   359.2 2644.37
   363.4 2643.73     367 2643.71   386.3  2644.8   401.6 2646.18   405.8  2647.4
   414.9 2651.61   420.6 2655.45   431.3 2664.23   435.5 2667.21   438.8 2668.98
#Mann= 4 ,-1,0
       0     .05       0   215.8      .1       0   275.7    .045       0
  293.58      .1       0
#XS Ineff= 2 , 0
        179.3537 2645.43315.2726         2645.43
Permanent Ineff=
       F       F
Bank Sta=275.7,293.58
XS Rating Curve= 0 ,0
Exp/Cntr(USF)=0,0
Exp/Cntr=0.3,0.1

Type RM Length L Ch R = 1 ,6069    ,118.3,117,116.4
XS GIS Cut Line= 4
2306331.66585597515342.894033167 2306262.6979061515601.907000472
2306290.28508605515672.4075714542306415.96001693515796.549881227
#Sta/Elev= 30
       0 2646.94      57 2645.56    97.6 2644.89   118.3 2644.78   172.1 2645.14
   242.4 2643.22     268 2642.79   297.3 2641.05   330.4 2642.06   380.1 2641.49
   385.2 2641.02   390.9 2638.82   396.5 2637.55   401.8 2637.43   407.5  2637.9
   413.9 2638.79   419.5 2639.37   430.5 2639.84   436.1  2641.1     439 2641.48
   447.6 2641.63     453 2641.99   458.8 2645.22   470.1 2655.66   475.7 2658.63
   481.3 2661.15   492.6 2660.76   498.2 2660.91   509.9 2663.28   520.4 2663.61
#Mann= 5 ,-1,0
       0     .05       0   390.9    .045       0   413.9     .05       0
  433.74      .1       0  473.74     .06       0
Bank Sta=390.9,413.9
XS Rating Curve= 0 ,0
Exp/Cntr(USF)=0,0
Exp/Cntr=0.3,0.1
